HEC-RAS study TETERCK.prj: TETERCK

--- TETERCK.g01 (geometry) --- (continued)

Type RM Length L Ch R = 1 ,43836.6 ,350.7,399.5,447.9
XS GIS Cut Line= 4
     1859745.294      236985.026     1859825.155      237280.165
     1860220.989       237295.79     1860398.072      237408.637
#Sta/Elev= 30
       0 1422.67    38.2 1420.01    95.6 1418.01   133.8 1415.55   152.9 1415.12
  223.321415.692   310.11414.778   344.4 1415.33   354.1 1413.91     359 1411.79
   373.4 1405.96     383 1406.06   392.7 1408.14   399.5 1411.05     412 1415.01
   421.7 1415.24  458.69 1413.54   566.6 1412.93   624.6 1413.35  664.051414.544
   701.9 1417.26   711.4 1416.78   730.5 1413.11   740.1 1413.33   749.6 1416.67
   768.7 1427.32   787.8 1435.17   816.4 1443.67   883.2 1460.93   911.9 1470.37
#Mann= 7 ,-1 , 0
       0     .12       0  223.32    .016       0   310.1     .12       0
     359    .045       0   399.5     .12       0  458.69     .06       0
  664.05     .12       0
#XS Ineff= 2 , 0
                          698.66         1418.24
Permanent Ineff=
       F       F
Bank Sta=359,399.5
XS Rating Curve= 0 ,0
Exp/Cntr=0.3,0.1

Type RM Length L Ch R = 1 ,43437   ,65,66,67.8
XS GIS Cut Line= 4
      1859692.33       237040.02     1859752.492      237075.682
     1859926.029      237721.764     1860009.196       237859.72
#Sta/Elev= 30
       0 1425.06    26.31420.754      35 1419.35    43.7 1418.46    52.4 1417.97
    69.9 1417.96   109.3 1415.76     129 1415.23  160.431415.363   178.2 1415.63
  208.821415.554   286.4 1414.52   355.2 1412.74   443.8 1409.83   483.1  1409.4
   601.2 1409.91     611 1408.84  614.74 1408.05   620.9 1406.92   630.7 1405.92
   640.5 1405.86   650.4 1406.64  656.18 1407.89     670 1410.51  676.691411.382
   719.2 1416.32   738.9 1419.56   757.9 1423.71   795.8 1433.05     900  1463.9
#Mann= 7 ,-1 , 0
       0     .12       0    26.3    .016       0  160.43     .12       0
  208.82    .016       0  614.74    .045       0  656.18    .016       0
  676.69     .12       0
Bank Sta=614.74,656.18
XS Rating Curve= 0 ,0
Exp/Cntr=0.3,0.1

Type RM Length L Ch R = 1 ,43371.1 ,71.7,56.2,39.1
XS GIS Cut Line= 4
     1859632.925      237058.736     1859693.087      237094.398
     1859866.624       237740.48     1859949.791      237878.436
#Sta/Elev= 30
       0 1435.15    26.2 1429.07    52.4 1422.28    69.9 1419.92    99.4 1417.56
   119.1 1416.28   138.8 1415.75  249.711415.203  261.941415.008   335.6 1414.61
   443.8 1411.85   473.3  1411.7     552 1412.98   571.7 1414.06   591.4 1415.94
     611 1416.51   620.9  1415.7   630.7 1413.13   640.5 1409.11   650.4 1406.38
   660.2 1405.95     670  1406.7   679.9  1408.6   689.7 1410.43   699.6 1411.61
   738.9 1414.85   776.8 1420.43   786.3 1422.61   862.1 1444.34     900 1457.09
#Mann= 5 ,-1 , 0
       0     .12       0  249.71     .06       0  261.94     .12       0
   640.5    .045       0   679.9     .12       0
Bank Sta=640.5,679.9
XS Rating Curve= 0 ,0
Exp/Cntr=0.3,0.1

Type RM Length L Ch R = 1 ,43314.8 ,449.2,452.2,455.4
XS GIS Cut Line= 3
     1859356.405       237483.29     1859724.461      237594.401
     1859943.211      237877.387
#Sta/Elev= 30
       0 1437.17    19.2 1428.93    38.4 1421.09    48.1 1417.78    61.71414.491
    76.9 1411.57    86.5 1410.49   105.7 1409.63   134.6 1409.77   182.6 1410.62
   240.3 1412.32   278.7 1413.11   384.5 1414.39  420.991414.015   481.1 1413.62
   490.8 1412.67  502.53 1408.97   510.1 1406.55   519.8 1405.85   529.5 1406.33
  545.03 1409.08   558.5 1410.85   577.8  1412.8   587.5 1414.22   606.8 1418.03
   626.1  1420.9   635.8 1423.08   703.5 1442.72   722.8 1448.95   742.1 1455.69
#Mann= 5 ,-1 , 0
       0     .12       0    61.7     .06       0  420.99     .12       0
  502.53    .045       0  545.03     .12       0
Bank Sta=502.53,545.03
XS Rating Curve= 0 ,0
Exp/Cntr=0.3,0.1

Type RM Length L Ch R = 1 ,42862.6 ,425.9,465.8,502.4
XS GIS Cut Line= 2
     1859212.308      237606.554     1859608.141      238212.456
#Sta/Elev= 30
       0 1441.74    39.1 1423.54    48.9 1419.43    58.7 1416.64   68.491415.521
   107.6 1414.38   136.9 1414.05   234.7 1414.47  264.151414.239   293.4 1413.69
   332.5 1412.37   352.1 1411.24   371.6  1409.8   381.4 1408.96  395.84 1407.33
     401 1406.67   410.8 1406.07   430.3 1407.02   440.1 1407.28   449.9 1407.64
   459.7  1408.4   469.4 1409.46     489 1412.18   508.6 1414.28   518.4 1415.87
   528.1 1418.42     577 1433.24   606.4 1441.73   655.3 1454.96   723.7 1472.53
#Mann= 5 ,-1 , 0
       0     .12       0   68.49     .06       0  264.15     .12       0
  395.84    .045       0   440.1     .12       0
Bank Sta=395.84,440.1
XS Rating Curve= 0 ,0
Exp/Cntr=0.3,0.1

Type RM Length L Ch R = 1 ,42396.9 ,449.2,422.3,395
XS GIS Cut Line= 4
     1859020.034      237669.488     1859069.947      237923.394
     1858976.631       238170.79     1859347.725      238300.998
#Sta/Elev= 30
       0 1446.95    47.9 1429.09    76.7 1417.98    86.3  1415.3    95.8 1413.92
   105.4 1413.32  141.04  1412.2  243.041411.471   268.6 1410.97   297.9 1409.63
   317.5 1408.01   329.6 1406.24   337.1 1405.15   346.9 1404.67   356.7 1405.02
   376.3 1406.47  445.021410.659   474.2 1411.61   523.2 1411.94   572.3 1413.01
   611.7 1413.96  624.231414.581   670.6 1418.38   700.2 1420.15   729.6 1420.73
     769 1420.31     828 1421.84   837.8 1422.77     887 1430.24   916.4 1435.48
#Mann= 7 ,-1 , 0
       0     .12       0  141.04     .06       0  243.04     .12       0
   329.6    .045       0   376.3     .12       0  445.02     .06       0
  624.23     .12       0
Bank Sta=329.6,376.3
XS Rating Curve= 0 ,0
Exp/Cntr=0.3,0.1

Type RM Length L Ch R = 1 ,41974.6 ,280.2,245.9,211.5
XS GIS Cut Line= 3
     1858594.687       237712.89     1858744.426      238116.536
      1859278.28      238287.977
#Sta/Elev= 30
       0 1448.68    19.6 1445.71    48.9 1440.27    58.7 1438.02    68.5 1435.24
   117.4 1418.96     137 1411.79   146.8 1408.76   156.6 1406.71     185 1402.22
   195.7 1401.43   205.5 1401.31     227 1401.89   244.6 1403.18   292.31407.609
   313.1 1409.04   342.5 1409.81   430.5 1409.01   499.4    1410   627.3 1411.01
   745.3 1413.66  770.741414.929   814.2 1418.67   843.7 1420.32   873.2 1420.78
   912.5 1420.33   961.7 1421.25   971.6 1421.52   981.4 1422.49   991.2 1423.99
#Mann= 5 ,-1 , 0
       0     .12       0     185    .045       0     227     .12       0
   292.3     .06       0  770.74     .12       0
Bank Sta=185,227
XS Rating Curve= 0 ,0
Exp/Cntr=0.3,0.1

Type RM Length L Ch R = 1 ,41728.7 ,384.3,333.6,277.9
XS GIS Cut Line= 2
     1858382.013       238018.88     1859228.367      238292.317
#Sta/Elev= 30
       0 1473.41     9.8 1466.83    19.6 1459.46    39.1 1443.39    48.9 1434.81
    68.4 1415.58    78.2 1407.72    87.2 1403.55      88 1403.18    97.7 1401.28
   107.5 1400.69   117.3 1401.22   129.4 1402.68   136.8 1403.48   166.2 1405.48
   185.7 1406.51  202.411406.973     303  1407.7   439.8  1409.5   557.1 1410.59
   635.3 1412.09   684.2 1413.37   703.7 1414.25   716.91415.265   762.4 1419.03
   772.1 1419.57   791.7 1420.32     821 1420.75   850.3 1420.42   889.4 1420.81
#Mann= 5 ,-1 , 0
       0     .12       0    87.2    .045       0   129.4     .12       0
  202.41     .06       0   716.9     .12       0
#XS Ineff= 2 , 0
                          204.33         1409.05
Permanent Ineff=
       F       F
Bank Sta=87.2,129.4
XS Rating Curve= 0 ,0
Exp/Cntr=0.3,0.1

Type RM Length L Ch R = 1 ,41395.2 ,390.7,402.3,417.5
XS GIS Cut Line= 4
     1858464.478      238442.057     1858562.135      238346.571
     1858657.621      238127.387     1859213.176      238307.508
#Sta/Elev= 30
       0 1458.67     9.8 1455.35    29.3 1449.22      39 1445.97    48.8 1442.47
    68.3 1434.95      78 1431.49    87.8 1428.24    97.6 1424.63   117.1 1416.34
   136.6 1408.55   146.1 1404.32  153.31 1402.14   155.7 1401.22   165.3 1400.36
     194 1402.04     280 1405.01   327.8  1406.3   375.7 1407.26   531.4 1409.16
     619 1410.05   716.3 1411.74     765 1413.15   784.5 1414.22  798.721415.362
   833.2 1418.11   852.6 1419.15   872.1 1419.83     911 1420.63   959.7 1420.64
#Mann= 4 ,-1 , 0
       0     .12       0  153.31    .045       0     194     .06       0
  798.72     .12       0
Bank Sta=153.31,194
XS Rating Curve= 0 ,0
Exp/Cntr=0.3,0.1

Type RM Length L Ch R = 1 ,40992.9 ,270.8,263.3,256.4
XS GIS Cut Line= 3
     1858768.298      238659.071     1859089.478      238368.272
     1859232.707      238344.401
#Sta/Elev= 30
       0 1438.77    28.9 1428.03    48.1 1421.15    67.4 1414.65    96.3 1405.25
   105.9 1402.01   115.5 1398.98   125.2 1396.95   134.8  1396.3   144.4 1397.06
  158.73 1398.93   163.7 1399.73   173.3  1400.9   182.9 1401.91  187.671402.323
   202.2 1403.53   231.1 1405.61   250.3 1406.89   298.5 1409.66  342.071411.868
   375.5 1413.53   404.4 1415.08   433.3 1416.38   462.3 1417.96   491.4 1419.31
   520.4 1420.52   530.1 1420.68   539.8 1420.62   568.8  1420.2   578.5 1420.25
#Mann= 5 ,-1 , 0
       0     .12       0   115.5    .045       0  158.73     .12       0
  187.67     .06       0  342.07     .12       0
Bank Sta=115.5,158.73
XS Rating Curve= 0 ,0
Exp/Cntr=0.3,0.1

Type RM Length L Ch R = 1 ,40729.6 ,273.7,270.3,266.7
XS GIS Cut Line= 3
     1858973.923       238851.14     1859226.527      238512.598
     1859304.652      238473.536
#Sta/Elev= 30
       0 1443.35    19.6 1433.18    58.9 1413.02    68.8 1407.86    78.6 1402.06
    88.4 1396.89    95.4  1394.9    98.2  1394.1   108.1 1393.72   117.9 1393.94
   147.4 1394.88   176.8 1396.03   186.6 1396.54   196.5 1397.17   206.3 1397.92
   225.9 1399.76     275 1404.82   294.7 1406.61   314.3 1408.14     334 1409.37
   343.8 1409.88   353.6 1410.33   363.5 1410.66   392.9  1411.5   402.8 1412.04
   412.6 1412.72   432.1 1415.08   451.5 1417.77   480.6 1421.43   509.7 1425.79
#Mann= 3 ,-1 , 0
       0     .12       0    95.4    .045       0   147.4     .12       0
Bank Sta=95.4,147.4
XS Rating Curve= 0 ,0
Exp/Cntr=0.3,0.1

Type RM Length L Ch R = 1 ,40459.3 ,546.8,593.5,636.9
XS GIS Cut Line= 3
     1859195.277      239023.015     1859367.152      238741.765
      1859434.86      238567.286
#Sta/Elev= 30
       0 1428.48     9.7 1426.74    19.4 1424.71    38.8 1420.21    58.2 1415.32
    77.6 1410.08    96.9 1404.66   106.6 1401.81   116.3 1398.17  119.82 1397.06
     126 1395.18   135.7 1394.22   145.4 1394.84   155.1 1396.14   164.8 1397.19
   174.5 1397.76   193.9 1398.16   203.6 1398.21   281.1 1397.87   310.2    1398
   319.9 1398.26     339 1399.09   348.3 1399.58   357.7 1400.31     367 1401.84
   385.8 1406.34   404.5  1410.5   441.9 1418.23     470 1423.56   516.8  1431.5
#Mann= 3 ,-1 , 0
       0     .12       0  119.82    .045       0   164.8     .12       0
Bank Sta=119.82,164.8
XS Rating Curve= 0 ,0
Exp/Cntr=0.3,0.1

Type RM Length L Ch R = 1 ,39865.9 ,653,676,702.7
XS GIS Cut Line= 3
     1859234.878      239062.717     1859955.364      239136.502
      1860055.19      239327.474
#Sta/Elev= 30
       0 1421.88    78.3 1404.49    88.1 1402.83   117.4 1400.62   195.7 1392.24
   225.1 1390.63   254.5  1390.3   342.6 1390.85   420.8 1393.45     460 1393.47
   489.4 1392.48   518.7 1390.45   528.5  1390.7  535.59 1392.33   538.3    1393
   548.1  1397.2   567.7 1406.54   577.4  1411.9   587.2 1418.36   616.6 1439.53
   626.4  1445.1   636.2 1449.25   694.9 1470.21   714.5  1476.6   724.2  1479.3
   763.4 1494.32     783  1502.6     832 1527.65     881 1553.85   939.7  1581.7
#Mann= 3 ,-1 , 0
       0     .12       0   489.4    .045       0  535.59     .12       0
Bank Sta=489.4,535.59
XS Rating Curve= 0 ,0
Exp/Cntr=0.3,0.1

Type RM Length L Ch R = 1 ,39189.8 ,832.9,836.7,838.8
XS GIS Cut Line= 2
     1859087.308      239257.595     1859691.475      239919.054
#Sta/Elev= 30
       0 1429.97    58.4 1406.08    68.2 1402.58    77.9  1400.4    87.6  1398.9
    97.4 1396.78   116.8 1391.51   126.6 1389.46   146.1 1387.15   175.3 1385.54
  201.031384.972   204.5 1384.94  245.27  1385.3     313 1386.54   389.5 1386.91
   507.91388.228   545.3 1388.23   584.2 1387.17   623.2 1384.97   632.9 1386.81
   642.7 1392.22   662.2 1407.79   681.6 1421.94   691.4 1428.52   710.8 1440.07
   720.6 1445.09     740 1453.85     818 1490.82   856.9 1510.52   895.8 1527.19
#Mann= 7 ,-1 , 0
       0     .12       0  201.03     .06       0  245.27     .12       0
     313     .06       0   507.9     .12       0   584.2    .045       0
   632.9     .12       0
Bank Sta=584.2,632.9
XS Rating Curve= 0 ,0
Exp/Cntr=0.3,0.1

Type RM Length L Ch R = 1 ,38353.1 ,325.9,322,318.2
XS GIS Cut Line= 3
     1858643.732      239499.783     1858668.037      239642.144
     1859261.787      240312.283
#Sta/Elev= 30
       0 1435.85    48.1  1419.1    86.6 1403.71   105.9 1397.02   115.5  1394.3
   144.4 1389.06   164.1 1384.25   183.8 1382.66   282.2 1381.52   311.7 1380.54
   321.5  1381.4   341.2  1383.8     351 1384.33  408.841385.803   577.3 1385.12
  657.421383.688   734.8 1384.63   744.6 1385.32   754.4  1386.8   764.3  1389.1
   803.6    1400   823.3 1406.45   833.1 1410.61     843 1415.73   872.5 1434.81
     902 1453.09   941.4 1476.91     961 1488.12   990.6 1503.22  1039.8  1526.6
#Mann= 5 ,-1 , 0
       0     .12       0   282.2    .045       0   321.5     .12       0
  408.84     .06       0  657.42     .12       0
#XS Ineff= 2 , 0
                          388.85         1388.65
Permanent Ineff=
       F       F
Bank Sta=282.2,321.5
XS Rating Curve= 0 ,0
Exp/Cntr=0.3,0.1

Type RM Length L Ch R = 1 ,38031.1 ,618.5,665.2,696.3
XS GIS Cut Line= 4
     1858429.146      239665.189      1858430.95      239766.217
     1858985.181      240289.103     1859186.856      240403.055
#Sta/Elev= 30
       0 1392.57    2.891392.259    36.7 1389.03    64.3 1387.17     101 1385.31
  135.621384.518   159.7 1383.97  177.921381.427   179.2 1381.23     189 1380.48
   198.7 1380.45   218.9 1380.77  382.781381.173  401.881381.064   501.6 1380.71
  735.471381.982   775.1 1382.72   794.6 1383.68   814.2  1387.4   872.6 1399.98
   882.3 1402.51     892 1406.45   901.6 1411.86   978.8 1460.96  1007.8 1478.85
  1046.4 1504.94  1065.7 1516.73  1075.3 1521.08    1085 1523.34  1094.6 1522.21
#Mann= 9 ,-1 , 0
       0    .016       0    2.89     .06       0  135.62    .016       0
  177.92     .12       0   179.2    .045       0   218.9     .06       0
  382.78     .12       0  401.88     .06       0  735.47     .12       0
#XS Ineff= 2 , 0
                          560.99         1386.22
Permanent Ineff=
       F       F
Bank Sta=179.2,218.9
XS Rating Curve= 0 ,0
Exp/Cntr=0.3,0.1

Type RM Length L Ch R = 1 ,37365.9 ,95.4,85.6,324.4
XS GIS Cut Line= 4
     1858218.069      239737.352      1858430.95      239914.151
      1858470.64      240832.424     1858665.479      240964.121
#Sta/Elev= 30
       0 1387.37    28.6 1386.27     124 1385.84  217.08 1383.01  251.821382.499
   306.1 1381.31   364.7 1381.85     531 1380.34   638.5 1380.89   658.1 1380.15
   671.9 1378.98   697.2 1377.34   717.5 1379.18   736.3 1380.45  772.71 1380.94
   853.6 1379.34  980.191379.695 1039.281380.598  1127.4  1381.8 1184.681385.063
 1203.431386.073  1225.2 1388.44  1244.8 1391.99 1251.091392.253  1254.6  1392.4
  1264.4 1391.34    1284 1387.13  1303.6 1385.65  1352.6 1386.54    1431 1386.79
#Mann= 11 ,-1 , 0
       0     .06       0  217.08     .12       0  251.82    .016       0
   671.9    .045       0   717.5     .12       0  772.71     .06       0
  980.19     .12       0 1039.28    .016       0 1184.68     .12       0
 1203.43    .016       0 1251.09     .12       0
Bank Sta=671.9,717.5
XS Rating Curve= 0 ,0
Exp/Cntr=0.3,0.1

Type RM Length L Ch R = 1 ,37280.3 ,713.7,669.6,139.2
XS GIS Cut Line= 4
     1858181.988      239757.197     1858371.416      239915.955
     1858411.105      240834.228     1858645.635      240991.183
#Sta/Elev= 30
       0 1389.13      19 1387.23      38 1386.39   161.6 1386.18   232.11383.537
   286.3 1382.13   364.5 1382.14   481.8 1380.53   648.1 1382.77   677.4  1381.4
   706.7 1377.55   726.3 1376.24   755.6  1377.3     7621377.535   843.6 1377.74
   941.4 1375.92  1000.1 1376.37  1009.8 1376.74  1058.7 1380.98  1078.3 1382.03
  1127.2 1383.79  1195.5 1383.89  1214.9 1384.79  1244.1 1387.02 1253.391387.181
  1283.1 1385.27 1293.831385.758  1312.3 1386.51 1378.441386.378  1448.5 1386.51
#Mann= 8 ,-1 , 0
       0     .06       0   232.1     .12       0   706.7    .045       0
   755.6     .06       0     762     .12       0 1253.39    .016       0
 1293.83     .12       0 1378.44     .06       0
Bank Sta=706.7,755.6
XS Rating Curve= 0 ,0
Exp/Cntr=0.3,0.1

Type RM Length L Ch R = 1 ,36610.7 ,529.5,522.6,761.8
XS GIS Cut Line= 4
      1857776.09      240472.956     1857949.701      240479.901
     1858368.104      240750.734     1858482.687      241156.984
#Sta/Elev= 30
       0 1494.27    19.3 1487.18      29 1482.52    77.2 1454.91    96.5 1445.38
   144.8 1429.17   154.4 1425.47   183.5  1411.8   222.6 1391.43   232.4 1386.85
   251.9 1379.45   271.5 1373.53   281.2  1371.8   320.3 1373.76     379 1376.32
   457.2 1377.51   476.7 1376.03   496.2 1373.41   515.8 1372.96   584.2 1376.58
   628.9 1379.61     682 1382.65   721.2 1383.88  791.761382.597   848.8 1382.38
   907.8 1385.79   996.1 1384.28 1054.741384.405 1085.291385.028  1094.3 1385.21
#Mann= 7 ,-1 , 0
       0     .12       0   271.5    .045       0   320.3     .12       0
   628.9     .06       0  791.76     .12       0 1054.74     .06       0
 1085.29     .12       0
Bank Sta=271.5,320.3
XS Rating Curve= 0 ,0
Exp/Cntr=0.3,0.1

Type RM Length L Ch R = 1 ,36088.2 ,662.2,664.2,666.2
XS GIS Cut Line= 3
     1857638.937      240924.345     1858350.743      241214.276
     1858416.715      241342.748
#Sta/Elev= 30
       0 1535.19    58.4 1509.21    68.1 1504.21    77.8 1498.46   136.2 1460.35
   175.1 1433.34   194.6 1418.99   233.5 1387.45   243.2  1380.6     253 1376.44
   272.4 1372.79   282.1 1371.73   291.9 1371.52   301.6 1371.59   321.1 1372.68
   369.7 1375.41   428.1 1377.19  470.751379.071  476.261379.265   496.2 1379.75
   525.4 1379.91   564.3 1378.71  585.311379.985   632.4 1381.49   749.1  1380.9
  781.571381.839  799.131382.444   864.9 1384.87  904.921387.173     913 1387.83
#Mann= 9 ,-1 , 0
       0     .12       0   272.4    .045       0   321.1     .12       0
  470.75     .06       0  476.26     .12       0  585.31     .06       0
  781.57     .12       0  799.13     .06       0  904.92     .12       0
#XS Ineff= 2 , 0
                          390.09         1378.85
Permanent Ineff=
       F       F
Bank Sta=272.4,321.1
XS Rating Curve= 0 ,0
Exp/Cntr=0.3,0.1

Type RM Length L Ch R = 1 ,35423.9 ,1976.7,1998,1992.4
XS GIS Cut Line= 3
     1857383.584      241266.649     1857418.307      241531.406
     1858138.793      241869.947
#Sta/Elev= 30
       0 1491.67    57.2 1467.17   162.1 1424.61   228.9 1399.14   296.5 1375.84
   306.3 1374.12   316.2 1373.67   424.3 1373.07   470.8 1371.12   493.1 1369.59
   502.9 1369.77   517.9 1371.09   532.4 1371.83  573.621370.554  644.641370.773
  646.921370.808   709.3 1373.01   748.6 1373.63  778.51 1375.29  778.621375.301
   807.6 1379.02     837 1385.18  858.621388.544   886.2 1391.46     896 1393.42
   910.41397.862  916.231399.731   945.2 1407.59  991.311417.495  1063.1 1432.26
#Mann= 12 ,-1 , 0
       0     .12       0   470.8    .045       0   517.9     .12       0
  573.62     .06       0  644.64     .12       0  646.92     .08       0
  778.51     .06       0  778.62     .12       0  858.62    .016       0
   910.4     .12       0  916.23     .06       0  991.31     .12       0
#XS Ineff= 2 , 0
                          718.27         1379.16
Permanent Ineff=
       F       F
Bank Sta=470.8,517.9
XS Rating Curve= 0 ,0
Exp/Cntr=0.3,0.1

Type RM Length L Ch R = 1 ,33426   ,952,994,973.2
XS GIS Cut Line= 2
     1856597.994      241861.267     1857717.786      242655.537
#Sta/Elev= 30
       0 1403.82    98.1  1406.1   176.5  1406.1   196.1 1405.83   235.4 1402.92
     255 1400.35   274.6 1395.48   343.2 1370.85   362.8 1369.05  395.241368.773
  428.491368.323   490.3 1367.74  551.341369.493  564.211369.637   576.4 1369.39
   598.2 1367.57   625.1 1368.54   663.91369.161  844.261368.833  894.151369.688
  956.161371.748    1010 1374.29 1104.331375.705  1127.7 1378.02  1147.3 1384.47
  1186.6 1401.84 1238.941428.366 1276.731440.571  1333.6 1465.68  1372.9 1481.46
#Mann= 14 ,-1 , 0
       0     .12       0  395.24     .06       0  428.49     .12       0
  551.34     .06       0  564.21     .12       0   576.4    .045       0
   625.1     .12       0   663.9     .08       0  844.26     .06       0
  894.15     .12       0  956.16     .06       0 1104.33     .12       0
 1238.94    .016       0 1276.73     .12       0
Bank Sta=576.4,625.1
XS Rating Curve= 0 ,0
Exp/Cntr=0.3,0.1

Type RM Length L Ch R = 1 ,32432   ,700.3,715.4,727.9
XS GIS Cut Line= 4
     1856308.932      242310.919     1856483.375      242293.447
     1856984.279      242989.739     1857626.727      242948.394
#Sta/Elev= 30
       0 1552.77    58.4 1539.53   107.1 1525.56   185.1    1510   204.6 1504.19
   253.3 1484.86   272.8  1475.5     341 1437.72   389.8 1412.32   399.5 1405.34
   428.7 1378.32   438.5 1372.63   448.2  1370.5   506.7 1367.48   526.2    1367
   565.2  1367.2   613.9  1368.9  787.881369.662  874.341371.248   896.6 1372.91
   925.8 1377.73   974.6 1381.41  1052.6 1381.75  1247.6  1388.3  1286.7 1394.78
 1419.261410.565 1427.381411.595 1489.261420.335 1636.581455.647  1676.8 1465.95
#Mann= 9 ,-1 , 0
       0     .12       0   506.7    .045       0   565.2     .06       0
  787.88     .12       0  874.34     .06       0 1419.26     .12       0
 1427.38    .016       0 1489.26     .12       0 1636.58    .016       0
Bank Sta=506.7,565.2
XS Rating Curve= 0 ,0
Exp/Cntr=0.3,0.1

Type RM Length L Ch R = 1 ,31716.6 ,1257.8,1353.5,1349.6
XS GIS Cut Line= 4
     1856236.015      242326.544     1855985.336      242460.345
     1856302.855      243349.982     1856283.845      243849.435
#Sta/Elev= 30
       0 1567.68    19.6 1566.67      49 1559.76     147 1526.52   284.2 1489.83
   343.2 1490.99   412.1 1489.51   461.3 1482.62   520.3 1461.25   549.8 1447.09
     599 1418.57   648.2 1382.52   658.1 1376.59   677.7 1372.22  726.491369.615
  772.341369.371   815.5 1370.01   835.2 1367.72   854.8 1365.32   884.4 1367.08
   982.8 1373.43  1110.7 1377.19  1218.9 1382.38 1396.711402.168 1440.341406.138
 1491.471414.617    1562 1428.08 1599.111437.757  1630.6 1446.98  1728.6  1470.8
#Mann= 9 ,-1 , 0
       0     .12       0  726.49     .06       0  772.34     .12       0
   835.2    .045       0   884.4     .06       0 1396.71    .016       0
 1440.34     .12       0 1491.47     .06       0 1599.11     .12       0
Bank Sta=835.2,884.4
XS Rating Curve= 0 ,0
Exp/Cntr=0.3,0.1

Type RM Length L Ch R = 1 ,30363.1 ,1264.9,1236.5,1196.6
XS GIS Cut Line= 3
     1854788.098      242425.503     1854829.765      242795.294
     1855647.473      243982.794
#Sta/Elev= 30
       0 1467.28   63.631447.152  138.641428.554  155.321424.198   215.4  1408.2
   254.6 1399.82   372.1 1379.07   429.51374.727   445.21373.142   499.6 1370.43
   656.6 1370.63   823.3 1366.07   901.8 1367.08  950.661365.986     990 1363.91
  1039.1    1364 1050.971364.428  1156.8  1367.6 1334.041367.005  1362.8 1369.18
    14061384.896  1441.2 1397.16  1505.31416.211 1543.181427.227  1578.5 1434.82
 1594.491441.164  1647.2 1468.74 1720.04 1498.36 1764.53 1515.61  1813.9  1533.4
#Mann= 17 ,-1 , 0
       0     .12       0   63.63     .06       0  138.64     .12       0
  155.32     .06       0   429.5     .12       0   445.2     .06       0
  950.66     .12       0     990    .045       0  1039.1     .12       0
 1050.97     .06       0 1334.04     .12       0    1406     .06       0
  1505.3     .12       0 1543.18    .016       0 1594.49     .12       0
 1720.04    .016       0 1764.53     .12       0
#XS Ineff= 2 , 0
          652.22 1379.16
Permanent Ineff=
       F       F
Bank Sta=990,1039.1
XS Rating Curve= 0 ,0
Exp/Cntr=0.3,0.1

Type RM Length L Ch R = 1 ,29126.6 ,719.2,719.2,724.6
XS GIS Cut Line= 4
     1854204.765      244133.836     1854574.557      243951.544
     1855168.307      243998.419     1855506.848      244128.628
#Sta/Elev= 30
       0 1571.31    49.1 1550.14   176.7 1492.12   196.3 1484.36   225.8 1476.14
  261.761462.265  305.25 1450.05   343.6 1439.42  413.831405.825  447.84  1397.7
   490.4 1382.19   529.4 1370.61     549 1368.49   656.4  1363.9     658  1363.9
   710.1 1363.91   861.4 1364.19   900.5 1368.73  936.331377.651   968.8 1384.41
   998.1 1399.42  1007.9 1402.41  1037.3 1406.95 1083.741416.511 1125.291422.056
 1162.881439.521  1194.1 1452.82 1214.751460.125  1341.2 1503.05  1370.6 1510.66
#Mann= 12 ,-1 , 0
       0     .12       0  261.76    .016       0  305.25     .12       0
  413.83    .016       0  447.84     .12       0     658    .045       0
   710.1     .06       0  936.33     .12       0 1083.74    .016       0
 1125.29     .12       0 1162.88    .016       0 1214.75     .12       0
Bank Sta=658,710.1
XS Rating Curve= 0 ,0
Exp/Cntr=0.3,0.1

Type RM Length L Ch R = 1 ,28407.4 ,477.1,495.8,514.5
XS GIS Cut Line= 2
     1854387.057      244493.211     1855241.223      244685.919
#Sta/Elev= 30
       0 1532.83   137.7 1473.44   177.1 1457.44   236.1 1434.35   265.6 1421.83
   275.5 1417.99   285.3 1415.07   324.7 1405.19  401.951383.214   413.2 1380.62
   432.9 1377.71  438.531376.532   452.6 1373.82   462.4 1372.65  525.161368.875
   541.1 1367.88     551 1367.12   570.6 1364.49   580.5 1363.95   590.3 1364.94
  596.81 1367.79   600.2 1369.08  610.461375.426   619.8  1379.6  648.421385.575
   718.2 1402.08   757.6 1412.28   806.8 1427.28   846.1 1440.58   875.6 1451.08
#Mann= 8 ,-1 , 0
       0     .12       0  401.95    .016       0  438.53     .06       0
  525.16     .12       0   541.1    .045       0  596.81     .12       0
  610.46    .016       0  648.42     .12       0
Bank Sta=541.1,596.81
XS Rating Curve= 0 ,0
Exp/Cntr=0.3,0.1

Type RM Length L Ch R = 1 ,27911.6 ,487.5,490.2,492.6
XS GIS Cut Line= 3
     1854413.098      244784.878     1854819.348      245139.044
     1855090.182      245113.003
#Sta/Elev= 30
       0 1483.38    29.4 1468.59    39.2 1464.14      49 1460.14   137.2 1427.49
   215.6 1400.26   225.4  1396.1     245 1386.02   264.6 1374.88  272.14 1369.94
   274.4 1368.62   284.2 1364.89     294 1363.89   303.8 1364.27   323.4 1368.16
   333.2 1369.76  344.361371.408   372.4 1375.35   389.41376.448   456.61379.988
  474.971380.874   529.2  1383.6   597.3 1387.61   636.1 1390.95   665.3 1394.15
   684.7 1396.65   713.9 1401.02   723.6 1403.02   762.4 1413.61     811 1428.05
#Mann= 7 ,-1 , 0
       0     .12       0  272.14    .045       0   333.2     .12       0
  344.36    .016       0   389.4     .12       0   456.6     .06       0
  474.97     .12       0
Bank Sta=272.14,333.2
XS Rating Curve= 0 ,0
Exp/Cntr=0.3,0.1

Type RM Length L Ch R = 1 ,27421.5 ,570.8,573.7,576.6
XS GIS Cut Line= 2
     1854163.098      245170.294     1854616.223      245623.419
#Sta/Elev= 30
       0 1446.07    77.7 1420.78   165.1 1392.98   194.2 1383.34   223.3 1374.61
     233 1372.11   242.7 1370.76   262.2  1369.7   281.6 1367.93   300.5 1365.88
   310.7 1364.69   320.4 1363.99   330.1 1363.91   339.8 1364.08   349.5 1364.88
   353.9 1365.47  380.821368.729  415.911372.583   427.2 1373.51   436.9 1374.79
   446.6 1376.88  457.091379.557   475.8 1384.58   514.6 1396.08   524.3 1398.81
   543.7 1403.68   563.1 1409.17   572.8 1411.31   582.6 1412.91   640.8 1421.16
#Mann= 6 ,-1 , 0
       0     .12       0   300.5    .045       0   353.9     .06       0
  380.82     .12       0  415.91    .016       0  457.09     .12       0
Bank Sta=300.5,353.9
XS Rating Curve= 0 ,0
Exp/Cntr=0.3,0.1

Type RM Length L Ch R = 1 ,26847.8 ,594.6,607.3,619.8
XS GIS Cut Line= 3
     1853798.515      245336.961      1853814.14      245597.378
      1854157.89      245998.419
#Sta/Elev= 30
       0 1467.04    38.6 1453.25    67.6 1443.49    77.3 1440.59   96.181436.045
   125.6 1429.39   144.9 1423.97   173.9 1415.04   183.6 1412.29   231.9 1399.88
   251.2 1395.46   309.8 1383.65   339.1 1376.95   348.9 1375.17   358.7 1373.83
     437 1364.81   446.7 1364.09   466.3 1363.91   485.9 1363.92   495.6 1364.26
   505.4 1365.85  543.891376.879   554.3 1379.66   573.9 1382.85  584.481385.101
   671.7 1410.31   730.4 1428.84   740.2 1432.24   759.7 1439.83   789.1 1450.31
#Mann= 6 ,-1 , 0
       0     .12       0   96.18     .06       0     437    .045       0
   495.6     .12       0  543.89    .016       0  584.48     .12       0
Bank Sta=437,495.6
XS Rating Curve= 0 ,0
Exp/Cntr=0.3,0.1

Type RM Length L Ch R = 1 ,26240.5 ,691.1,645.3,599.6
XS GIS Cut Line= 3
     1853082.369      245756.232     1853342.786      245803.107
     1853566.744      246370.815
#Sta/Elev= 30
       0 1468.32    29.4 1457.33    78.4 1438.25    88.2 1434.68      98 1431.57
  126.111423.595   186.2 1407.01   264.6 1386.47     284 1383.26   303.4 1380.98
   332.4 1378.57   400.2 1372.28   458.3 1369.13  523.391366.306   535.8 1365.78
   574.6 1363.86   584.3 1364.06     594 1365.81   632.7 1380.96  644.411385.848
   652.1 1388.94   661.8 1391.95   671.5 1394.06   681.2 1396.81  691.151400.799
  717.321412.018     749 1425.42   758.6 1429.01  774.021434.182   874.9  1468.1
#Mann= 9 ,-1 , 0
       0     .12       0  126.11     .06       0  523.39     .12       0
   535.8    .045       0     594     .12       0  644.41    .016       0
  691.15     .12       0  717.32     .06       0  774.02     .12       0
Bank Sta=535.8,594
XS Rating Curve= 0 ,0
Exp/Cntr=0.3,0.1

Type RM Length L Ch R = 1 ,25595.2 ,713.4,732.4,750.8
XS GIS Cut Line= 3
      1852720.39      246352.586     1852918.307      246461.961
     1853486.015      246456.753
#Sta/Elev= 30
       0 1471.45    49.2 1447.71    88.5 1430.48    98.3 1427.14   196.6 1399.75
   206.5  1397.3   235.9 1392.73   245.7 1390.39   255.5 1387.21   275.1 1379.31
   294.6 1368.75   304.4 1364.96   314.2 1364.14   353.4 1367.49   431.7 1372.78
   481.81376.931  511.341377.739   529.6  1377.8  543.331378.949   568.7 1383.41
   578.5 1383.92   607.9 1382.65   617.7 1383.03   627.5 1384.94   637.2  1389.2
  669.971407.751   715.6    1431  736.271437.993   754.7 1443.88   793.9  1457.8
#Mann= 8 ,-1 , 0
       0     .12       0   294.6    .045       0   353.4     .06       0
   481.8     .12       0  511.34    .016       0  543.33     .12       0
  669.97     .06       0  736.27     .12       0
Bank Sta=294.6,353.4
XS Rating Curve= 0 ,0
Exp/Cntr=0.3,0.1

Type RM Length L Ch R = 1 ,24862.8 ,576.4,577.5,578.5
XS GIS Cut Line= 2
     1852366.223      246915.086     1852998.168      247241.475
#Sta/Elev= 30
       0 1464.89   25.921454.572    68.2 1437.75      78 1434.23    87.7 1431.15
   116.9 1424.44   126.7 1421.76   136.4 1418.71   155.9 1413.59   194.9 1404.84
   243.6 1392.65     302 1378.78   311.8 1376.55   321.5 1374.88  331.681373.858
   350.8 1372.04   360.5 1370.62   389.7 1365.24   403.6 1363.63     419 1362.36
   428.7 1361.86   438.4    1362   459.1 1363.82   477.4 1365.17   487.2 1367.29
   496.3 1370.62   535.9 1387.57   604.1 1418.02   672.3 1446.57   711.2 1463.31
#Mann= 6 ,-1 , 0
       0     .12       0   25.92     .06       0  331.68     .12       0
   403.6    .045       0   459.1    .016       0   496.3     .12       0
Bank Sta=403.6,459.1
XS Rating Curve= 0 ,0
Exp/Cntr=0.3,0.1

Type RM Length L Ch R = 1 ,24285.3 ,153.8,160.6,168
XS GIS Cut Line= 3
     1851956.397      247474.723     1852296.762      247513.681
     1852776.554      247778.181
#Sta/Elev= 30
       0 1384.17    48.9 1382.89   117.5 1382.44  158.961382.921   169.41382.805
   215.3 1381.06   313.2 1373.75     3421373.386  386.441372.553  456.021371.029
  496.491369.773   538.3 1367.65  573.19 1364.15   606.7 1359.52   616.5 1360.37
   626.3 1363.12  634.451365.706   655.7    1370   665.4 1373.04  672.08 1375.91
     685 1380.41   704.6 1386.07   714.4 1390.77   724.1 1396.64   753.5 1416.33
   763.3 1421.91   782.8 1431.47   812.2 1444.85     822 1450.42   890.5 1494.64
#Mann= 11 ,-1 , 0
       0     .12       0  158.96     .06       0   169.4     .12       0
     342    .016       0  386.44     .12       0  456.02     .06       0
  496.49     .12       0  573.19    .045       0   626.3     .12       0
  634.45    .016       0  672.08     .12       0
Bank Sta=573.19,626.3
XS Rating Curve= 0 ,0
Exp/Cntr=0.3,0.1

Type RM Length L Ch R = 1 ,24124.7 ,132.3,132.3,132.3
XS GIS Cut Line= 4
     1851942.456      247500.761     1852286.922      247644.288
     1852532.969      247845.227     1852740.059      247869.831
#Sta/Elev= 30
       0 1386.68    88.4  1384.4   117.8 1382.82  168.641381.915  172.561381.759
   235.7 1378.62   255.3 1377.12   284.8 1373.98  308.06 1373.11   324.1 1373.22
  344.781372.641  411.04 1369.74   430.9 1368.57  454.261367.933  467.341367.438
   517.6 1365.23   556.1 1362.93   594.6 1359.44   604.2 1359.59   613.8 1361.43
   633.1 1366.52  641.621368.242   671.6 1373.14  689.41 1378.42   719.3  1388.3
   728.8 1392.12   738.2 1397.23   785.6 1426.77     833 1454.97   899.4 1496.85
#Mann= 12 ,-1 , 0
       0     .12       0  168.64     .06       0  172.56     .12       0
  308.06    .016       0  344.78     .06       0  411.04     .12       0
  454.26     .06       0  467.34     .12       0   556.1    .045       0
   613.8     .12       0  641.62    .016       0  689.41     .12       0
#XS Ineff= 2 , 0
          527.35 1373.24
Permanent Ineff=
       F       F
Bank Sta=556.1,613.8
XS Rating Curve= 0 ,0
Exp/Cntr=0.3,0.1

Type RM Length L Ch R = 1 ,23992.4 ,190.2,179.5,168.1
XS GIS Cut Line= 4
     1851878.482      247612.099     1852222.948      247755.627
     1852468.995      247956.565     1852676.085       247981.17
#Sta/Elev= 30
       0  1395.2    68.7  1392.2   117.8 1387.69  177.061383.543     216 1381.05
   245.61378.147  289.581373.277   324.1 1371.99   382.8 1373.46   450.2 1373.18
  557.091366.193     585 1363.86   613.8 1359.11   623.5 1360.67   633.1 1363.48
   645.8 1367.22     662 1370.18   681.2 1372.32  701.081373.245   728.8 1373.72
  735.311374.606   757.2  1380.1   766.7 1383.36   776.2    1388   785.6 1395.24
   804.6 1411.46   814.1  1417.4     833 1427.16     871 1443.54   899.4  1458.4
#Mann= 9 ,-1 , 0
       0     .12       0  177.06     .06       0   245.6     .12       0
  289.58     .06       0  557.09     .12       0     585    .045       0
   633.1     .12       0  701.08    .016       0  735.31     .12       0
#XS Ineff= 2 , 0
          560.37 1371.62
Permanent Ineff=
       F       F
Bank Sta=585,633.1
XS Rating Curve= 0 ,0
Exp/Cntr=0.3,0.1

Type RM Length L Ch R = 1 ,23812.9 ,456.8,411,365.2
XS GIS Cut Line= 4
     1851942.044      248198.512      1852235.25      248030.379
     1852561.263      248167.756     1852694.538       248085.74
#Sta/Elev= 30
       0  1406.2   91.321390.193   106.2 1387.81  117.851387.431   144.8 1388.28
   154.5 1387.02  163.431384.857  174.461382.445   193.1 1380.62     280  1375.7
     338 1374.13   387.1 1371.44   406.8  1369.8   416.6 1368.44   426.4 1365.65
   436.3 1361.69   446.1 1358.67   455.9 1357.81   465.7 1358.47   495.2 1362.39
   524.7 1365.92   544.4 1367.58   583.7 1367.82  672.881371.549   701.6 1372.43
   711.3 1373.24   721.1 1376.28  726.331378.628   799.4 1413.71   848.3 1443.32
#Mann= 9 ,-1 , 0
       0     .12       0   91.32     .06       0  117.85    .016       0
  163.43     .06       0  174.46     .12       0   436.3    .045       0
   495.2     .12       0  672.88    .016       0  726.33     .12       0
#XS Ineff= 2 , 0
                          537.67         1371.62
Permanent Ineff=
       F       F
Bank Sta=436.3,495.2
XS Rating Curve= 0 ,0
Exp/Cntr=0.3,0.1

Type RM Length L Ch R = 1 ,23401.9 ,369.9,402.2,434.1
XS GIS Cut Line= 2
     1852290.611      248631.145     1852737.597      248159.554
#Sta/Elev= 30
       0 1414.67     9.7 1411.87    19.4 1409.84   51.341407.021    67.9 1404.18
    87.3 1400.36   126.1 1391.81   174.6 1379.95   203.7 1372.02   213.4 1370.26
     278 1362.92   300.6 1358.35   310.3 1358.38   329.7 1361.68   334.6 1362.22
  396.811368.165   436.4    1371  476.281372.736   504.3 1373.97  511.641375.279
     514  1375.7   533.4  1382.1   552.8    1387  562.351389.796   572.2 1393.11
   591.6 1400.55     611 1409.27   630.4 1419.06   640.1 1424.88   649.8 1431.18
#Mann= 8 ,-1 , 0
       0    .016       0   51.34     .12       0     278    .045       0
   334.6     .12       0  396.81     .06       0  476.28    .016       0
  511.64     .08       0  562.35     .12       0
Bank Sta=278,334.6
XS Rating Curve= 0 ,0
Exp/Cntr=0.3,0.1

Type RM Length L Ch R = 1 ,22999.7 ,498.4,512.5,526.1
XS GIS Cut Line= 2
     1852366.476      248719.311     1853092.315      248739.815
#Sta/Elev= 30
       0 1414.74    98.1 1413.32   107.9 1412.88   117.8 1411.66   127.6 1409.55
   166.8  1398.8   186.4 1393.72   215.9 1386.99   264.9 1376.53   284.6 1371.84
   294.4 1368.84  311.31 1361.44     314 1360.24   323.8 1357.95   333.6 1357.65
   343.4 1358.02   353.2 1359.01   372.9 1361.49   392.5 1363.85  431.791367.449
  475.62 1372.41  506.641374.984   529.9 1376.65   549.5 1377.32  560.641378.008
   569.1 1379.07   618.2 1386.65   637.8 1390.55   667.2 1397.91   726.1 1413.92
#Mann= 7 ,-1 , 0
       0     .12       0  311.31    .045       0   372.9     .12       0
  431.79    .016       0  475.62     .06       0  506.64    .016       0
  560.64     .12       0
Bank Sta=311.31,372.9
XS Rating Curve= 0 ,0
Exp/Cntr=0.3,0.1

Type RM Length L Ch R = 1 ,22487.2 ,497.3,490.8,483.3
XS GIS Cut Line= 3
      1852442.34      249039.173     1852920.082       249236.01
     1853299.404       249285.22
#Sta/Elev= 30
       0 1402.11      39  1391.8   146.2 1374.88     273 1366.25   331.5 1365.46
   380.2 1366.36     390 1365.86   405.6 1361.86   419.2 1358.48   438.7 1357.36
   448.5 1359.18  453.75 1361.45   487.5 1380.06   497.2 1384.25  501.941385.077
   516.7 1386.78  533.171390.807   555.9 1398.33   585.4  1404.1   595.2 1407.22
     605 1411.88   624.6 1424.47   644.2 1434.95  714.571464.121   742.3 1473.26
  755.371479.879   781.5 1496.97   801.1 1508.71   879.6 1545.31   899.2 1552.88
#Mann= 7 ,-1 , 0
       0     .12       0   405.6    .045       0  453.75     .12       0
  501.94    .016       0  533.17     .12       0  714.57    .016       0
  755.37     .12       0
Bank Sta=405.6,453.75
XS Rating Curve= 0 ,0
Exp/Cntr=0.3,0.1

Type RM Length L Ch R = 1 ,21996.4 ,245.4,278.6,311.8
XS GIS Cut Line= 3
     1852224.999      249377.487     1853057.458       249549.72
     1853419.262      249516.102
#Sta/Elev= 30
       0 1417.53    32.31418.277    87.9 1422.99    97.7 1421.12   117.2 1412.15
   166.1 1385.29   195.4 1361.79     207 1355.59     215  1353.6   244.3  1352.9
   264.7 1355.35  265.271355.491   283.4 1358.85   371.3 1361.05  441.681366.339
  530.221369.507  537.631369.584   566.7 1370.84  601.391379.449  617.211381.617
  663.111395.761  700.771403.437  788.951437.592     811 1443.34  827.531451.017
   869.7 1461.03  945.091500.474   977.8 1515.53  1105.4 1547.44  1213.4 1577.25
#Mann= 15 ,-1 , 0
       0    .016       0    32.3     .12       0     207    .045       0
   264.7     .04       0  265.27     .06       0  441.68    .016       0
  530.22     .06       0  537.63     .12       0  601.39    .016       0
  617.21     .12       0  663.11    .016       0  700.77     .12       0
  788.95    .016       0  827.53     .12       0  945.09     .06       0
Bank Sta=207,264.7
XS Rating Curve= 0 ,0
Exp/Cntr=0.3,0.1

Type RM Length L Ch R = 1 ,21717.9 ,278.8,287.2,295.7
XS GIS Cut Line= 3
     1852190.142      249422.596     1852633.027      250255.055
      1852486.97      250568.185
#Sta/Elev= 30
       0 1417.17     9.8 1413.37    19.6 1412.17   33.591412.496    68.8 1416.02
    78.6 1415.35    88.4  1412.8     167 1379.92   196.4 1361.93   206.3 1356.35
   212.7 1354.03   225.9 1352.24   255.4 1352.51     275 1354.25  279.291354.872
  312.461358.784  395.711364.388   481.3 1368.57   628.6 1372.34   785.8 1374.94
   893.8  1369.1   990.9 1368.26  1029.3 1371.42 1048.021375.388  1087.51383.131
  1144.5  1396.1  1173.3 1403.73  1211.7 1414.78  1259.7  1430.7  1288.5  1439.1
#Mann= 9 ,-1 , 0
       0    .016       0   33.59     .12       0   212.7    .045       0
     275     .04       0  279.29     .06       0  312.46     .12       0
  395.71     .06       0 1048.02    .016       0  1087.5     .12       0
Bank Sta=212.7,275
XS Rating Curve= 0 ,0
Exp/Cntr=0.3,0.1

Type RM Length L Ch R = 1 ,21430.6 ,392.8,375.2,357.7
XS GIS Cut Line= 4
       1852002.1      249556.405     1852101.927      249920.989
     1852097.586      249923.159     1852095.416       250417.95
#Sta/Elev= 30
       0  1420.3    53.21399.426    67.8 1395.58    87.2 1393.38   97.411390.269
   164.8 1361.35   193.8 1354.34   213.2 1351.42   222.9  1351.2   271.4 1351.32
   281.1 1352.18  304.771357.598   319.8 1360.73  335.261362.146     378 1364.46
  423.541364.787   460.5 1365.88  487.051368.421  516.591370.484  549.521372.157
  569.331374.782   615.7 1382.85   644.8 1389.23   664.2 1390.96  685.971391.107
     703  1391.3  728.43 1393.88  763.161398.305   858.2 1416.03   877.6 1422.11
#Mann= 15 ,-1 , 0
       0     .12       0    53.2    .016       0   97.41     .12       0
   213.2    .045       0   271.4     .04       0  304.77     .12       0
  335.26     .06       0  423.54    .016       0  487.05     .06       0
  516.59     .12       0  549.52     .06       0  569.33     .12       0
  685.97    .016       0  728.43     .12       0  763.16     .06       0
Bank Sta=213.2,271.4
XS Rating Curve= 0 ,0
Exp/Cntr=0.3,0.1

Type RM Length L Ch R = 1 ,21055.4 ,561,548,534.9
XS GIS Cut Line= 3
     1851597.586      249817.256     1851994.722      250259.964
     1851996.892      250418.384
#Sta/Elev= 30
       0 1384.53    29.2 1373.37      39    1370    48.8 1368.47    58.5 1368.37
   81.211369.989    97.5 1370.88   107.2 1370.62     117 1369.02   122.61367.523
   165.8 1354.88   175.5  1352.5   185.2 1351.29     195 1351.21   247.5 1351.56
   253.5  1351.9  280.781358.212   292.5 1359.46   321.7 1360.21   399.7 1364.16
   458.2 1367.68     468 1368.74   477.7 1370.51  533.051383.666     546 1386.39
   555.7 1387.96  574.651389.755  615.651395.237     660 1401.89   753.2 1420.21
#Mann= 9 ,-1 , 0
       0     .12       0   81.21    .016       0   122.6     .12       0
   185.2    .045       0   247.5     .04       0  280.78     .06       0
  533.05    .016       0  574.65     .12       0  615.65     .06       0
Bank Sta=185.2,247.5
XS Rating Curve= 0 ,0
Exp/Cntr=0.3,0.1

Type RM Length L Ch R = 1 ,20507.4 ,399.2,379.7,360
XS GIS Cut Line= 3
     1851202.187      250292.516     1851506.875      250456.579
     1851756.875      250677.933
#Sta/Elev= 30
       0 1368.06   30.581368.531   31.781368.553    57.7 1368.67    67.3 1367.52
   78.111364.373    86.5 1361.27    96.1 1358.64   105.7 1357.47   153.8 1355.51
   163.4 1353.83   182.6 1348.32  186.15 1347.81   201.9 1346.66   230.7 1346.54
   240.3 1346.76   249.9 1347.86   256.6 1349.04  305.181358.001   336.4 1363.65
  407.921378.489   434.4 1382.48  453.391388.253  483.011397.658  495.85  1400.8
   522.8  1406.8   542.5 1412.98   562.1 1421.32     621 1448.17     680 1471.62
#Mann= 12 ,-1 , 0
       0     .06       0   30.58     .12       0   31.78    .016       0
   78.11     .12       0  186.15    .045       0   249.9     .04       0
   256.6     .12       0  305.18     .06       0  407.92    .016       0
  453.39     .12       0  483.01     .06       0  495.85     .12       0
Bank Sta=186.15,249.9
XS Rating Curve= 0 ,0
Exp/Cntr=0.3,0.1

Type RM Length L Ch R = 1 ,20127.7 ,291.5,302.7,313.2
XS GIS Cut Line= 3
     1851017.291      250745.641     1851564.262      250730.972
     1851699.583      250776.891
#Sta/Elev= 30
       0  1365.6   12.321366.108    38.11367.312    58.6 1367.52   80.351366.904
    97.7 1365.98   107.5 1364.72   156.3 1355.88   175.9 1351.81   205.2 1343.81
     215 1342.65   224.7  1342.5   273.6 1343.56  278.151343.834  307.681346.127
   322.4 1348.26  427.451368.409   439.7 1369.97   449.5 1372.21  455.371374.564
   478.8 1385.35   508.1 1400.16   527.6 1408.99   556.7 1419.08   585.3 1425.41
   594.8 1428.63   623.4 1442.52     652 1458.42   661.5 1463.16   690.1 1475.46
#Mann= 10 ,-1 , 0
       0     .06       0   12.32     .12       0    38.1    .016       0
   80.35     .12       0   205.2    .045       0   273.6     .04       0
  278.15     .12       0  307.68     .06       0  427.45    .016       0
  455.37     .12       0
Bank Sta=205.2,273.6
XS Rating Curve= 0 ,0
Exp/Cntr=0.3,0.1

Type RM Length L Ch R = 1 ,19825   ,370.1,377.4,383.9
XS GIS Cut Line= 3
     1850996.458      250966.995      1851410.52       251076.37
     1851569.375       251076.37
#Sta/Elev= 30
       0 1365.59   39.371364.823    97.3 1362.83   116.8 1361.22     146 1357.64
   204.4 1349.73   243.3 1341.81  249.291340.997   253.9 1340.44   262.8 1339.95
   311.5  1339.8   321.2 1340.01   330.9 1341.61   340.7 1344.78  345.121345.928
   350.4  1347.3   360.1 1348.17   379.6 1348.41   389.3 1348.94   399.1 1349.84
   408.8 1351.14   418.5 1352.79  454.791359.759   484.3 1364.42  495.931368.113
   512.4 1374.93   521.7 1379.53   549.7 1394.26   568.4 1403.58   587.1 1412.44
#Mann= 8 ,-1 , 0
       0    .016       0   39.37     .12       0  249.29     .04       0
   253.9    .045       0   321.2     .04       0  345.12     .12       0
  454.79    .016       0  495.93     .12       0
Bank Sta=253.9,321.2
XS Rating Curve= 0 ,0
Exp/Cntr=0.3,0.1

Type RM Length L Ch R = 1 ,19447.6 ,335.5,337.4,338.7
XS GIS Cut Line= 3
     1850899.236       251255.19     1851284.652      251435.745
     1851447.847      251456.579
#Sta/Elev= 30
       0 1373.92   31.691364.163    38.7 1362.32    48.4 1361.07      58  1360.4
   68.631358.925   106.4 1351.24   116.1 1349.48   125.8  1348.1   135.4 1347.02
   193.5 1340.78   212.8 1338.95   270.8  1335.1   280.5 1334.56   299.9 1333.98
   357.9 1333.05   367.6 1333.72   377.2 1337.03   386.9 1342.77  388.341343.426
   396.6 1347.19   406.3 1347.72   415.9 1347.36   425.6 1347.46  435.391347.864
     474 1349.82   493.4  1351.2  507.781352.548  540.251355.533   590.1 1359.96
#Mann= 9 ,-1 , 0
       0     .12       0   31.69    .016       0   68.63     .12       0
   299.9    .045       0   367.6     .04       0  388.34    .016       0
  435.39     .06       0  507.78    .016       0  540.25     .06       0
Bank Sta=299.9,367.6
XS Rating Curve= 0 ,0
Exp/Cntr=0.3,0.1

Type RM Length L Ch R = 1 ,19110.2 ,423.5,423.5,423.9
XS GIS Cut Line= 3
     1850788.125      251557.273     1851180.486      251762.134
     1851364.513      251807.273
#Sta/Elev= 30
       0 1401.77    19.7 1391.89    29.5 1386.49    68.8 1360.47   78.781354.477
    88.5 1350.52   108.2 1347.97  113.551346.731   137.7 1340.31   147.5 1338.59
   196.7  1336.5   206.6  1335.4   236.1 1329.22   245.9 1328.03   314.8 1327.54
   324.6 1328.49   334.4    1331  347.891335.335   354.1 1337.16   363.9  1338.8
   373.8 1339.71  389.111341.923   413.1 1344.56   442.6 1345.69   461.6 1345.78
   508.9 1344.54  541.261344.425   584.7 1346.55  624.181350.493   632.1 1351.36
#Mann= 9 ,-1 , 0
       0     .12       0   78.78    .016       0  113.55     .12       0
   245.9    .045       0   324.6     .04       0  347.89    .016       0
  389.11     .06       0  541.26     .12       0  624.18     .06       0
Bank Sta=245.9,324.6
XS Rating Curve= 0 ,0
Exp/Cntr=0.3,0.1

Type RM Length L Ch R = 1 ,18686.8 ,548.7,556.2,563
XS GIS Cut Line= 4
     1850666.597      251956.579     1850777.708      252026.023
     1851034.652       252161.44     1851177.013      252272.551
#Sta/Elev= 30
       0 1381.38     9.4 1375.63    28.1 1362.94    37.4 1357.45    46.8 1352.92
    56.2 1348.96   65.361345.769    74.9 1343.79   96.291342.212   140.7 1336.56
   189.1 1328.62   208.5 1325.89   218.2 1325.26   232.6 1325.08   266.6 1324.53
   292.9 1325.19   334.3 1326.72     344 1327.74   363.4 1330.84   373.1 1331.98
   392.4 1333.65   411.8 1334.78   440.5  1335.5  528.961335.577   535.5 1335.68
     545 1336.84   554.5 1340.04     564 1344.24   573.6 1348.09   602.1 1358.07
#Mann= 6 ,-1 , 0
       0     .12       0   65.36    .016       0   96.29     .12       0
   232.6    .045       0   292.9     .06       0  528.96     .12       0
Bank Sta=232.6,292.9
XS Rating Curve= 0 ,0
Exp/Cntr=0.3,0.1

Type RM Length L Ch R = 1 ,18130.6 ,501.3,505.6,509.1
XS GIS Cut Line= 3
     1850427.013      252407.968     1850777.708      252689.218
     1850867.986      252730.884
#Sta/Elev= 30
       0 1331.72     9.8 1328.82   12.791328.719   16.021328.611    19.6 1328.49
    39.1  1334.5    48.9 1335.19   62.281333.143    78.2 1329.18   89.541327.428
   117.3 1326.03  138.691325.948   185.7  1327.5   195.4 1326.83     215 1320.46
   224.8 1318.33  234.561317.629     235 1317.62   295.7 1317.63  298.91 1317.74
   332.3 1319.76     342 1319.15   371.4 1315.37   381.1 1315.16   390.9 1316.24
   410.4 1322.71  437.091337.636   449.5 1342.84  456.641345.037     549 1371.41
#Mann= 12 ,-1 , 0
       0     .12       0   12.79     .06       0   16.02    .016       0
   62.28     .12       0   89.54     .06       0  138.69     .12       0
  234.56     .04       0     235    .045       0   295.7     .04       0
  298.91     .12       0  437.09     .06       0  456.64     .12       0
Bank Sta=235,295.7
XS Rating Curve= 0 ,0
Exp/Cntr=0.3,0.1
